--- 25_ras.prj (project) ---

Proj Title=25
Current Plan=p01
Default Exp/Contr=0.3,0.1
English Units
Geom File=g01
Flow File=f01
Plan File=p01
Y Axis Title=Elevation
X Axis Title(PF)=Main Channel Distance
X Axis Title(XS)=Station
BEGIN DESCRIPTION:
RFD model 25 exported to HEC-RAS
END DESCRIPTION:

--- 25_ras.p01 (plan) ---

Plan Title=Plan 01
Program Version=4.10
Short Identifier=Plan 01
Geom File=g01
Flow File=f01
Subcritical Flow
Calc Critical at every XS
Secant Critical Depth

--- 25_ras.f01 (steady flow) ---

Flow Title=Flow 01
Program Version=5.01
Number of Profiles= 5
Profile Names=10yr,25yr,50yr,100yr,500yr
River Rch & RM=25,49,4192.087
   97.42  172.36  243.96  328.93  574.88
River Rch & RM=25,49,4049.834
  101.18  179.16  253.78  342.47  599.92
River Rch & RM=25,49,3907.581
  109.93  195.01  276.72  374.12  658.68
River Rch & RM=25,49,3765.328
  153.41  274.14  391.74  533.64  958.75
River Rch & RM=25,49,3623.075
  157.12  280.92  401.62   547.4   984.9
River Rch & RM=25,49,3480.821
  192.23  345.21  495.64  678.63 1236.07
River Rch & RM=25,49,3336.905
  198.36  356.48  512.16  701.75 1280.62
River Rch & RM=25,49,3240.406
   209.4  376.76  541.91  743.43 1361.15
River Rch & RM=25,49,2939.559
  227.76  410.54  591.54  813.06 1496.26
River Rch & RM=25,49,2829.319
  232.03  418.42  603.13  829.34 1527.94
River Rch & RM=25,49,2752.672
  232.64  419.55  604.78  831.67 1532.47
River Rch & RM=25,49,2593.389
  238.14  429.68  619.69  852.61  1573.3
River Rch & RM=25,49,2444.841
  278.93  505.03  730.78 1009.07 1879.97
River Rch & RM=25,49,2298.682
  280.75   508.4  735.76  1016.1 1893.81
River Rch & RM=25,49,2159.189
  309.86  562.33   815.5 1128.73 2116.38
River Rch & RM=25,49,1959.723
  323.18  587.03  852.07 1180.48 2219.08
River Rch & RM=25,49,1860.604
  329.83  599.38  870.37 1206.39 2270.58
River Rch & RM=25,49,1761.486
  415.36  758.63 1106.97 1542.37 2943.89
River Rch & RM=25,49,1662.367
  423.16   773.2 1128.67 1573.26 3006.25
River Rch & RM=25,49, 1464.13
  444.14  812.41 1187.11 1656.53 3174.69
River Rch & RM=25,49,1365.011
  451.93  826.97 1208.82  1687.5 3237.45
River Rch & RM=25,49,1166.774
  462.11     846 1237.23 1728.02 3319.68
River Rch & RM=25,49,1067.655
  483.04  885.18 1295.73 1811.55 3489.53
River Rch & RM=25,49,968.5368
  486.03  890.78 1304.09  1823.5 3513.85
River Rch & RM=25,49,869.4181
  494.39  906.45 1327.51 1856.95 3582.03
River Rch & RM=25,49,744.8112
  497.98  913.16 1337.54  1871.3 3611.29
River Rch & RM=25,49,467.5351
  502.16     921 1349.25 1888.04 3645.45
River Rch & RM=25,49,271.1879
  540.92  993.71 1458.05 2043.72  3963.9
River Rch & RM=25,49,140.0477
  546.28 1003.77 1473.12 2065.31 4008.17
River Rch & RM=25,49,       0
  547.47 1006.01 1476.47  2070.1 4018.01
Boundary for River Rch & Prof#=25,49,1
Up Type= 0
Dn Type= 2
Boundary for River Rch & Prof#=25,49,2
Up Type= 0
Dn Type= 2
Boundary for River Rch & Prof#=25,49,2
Up Type= 0
Dn Type= 2
Boundary for River Rch & Prof#=25,49,2
Up Type= 0
Dn Type= 2
Boundary for River Rch & Prof#=25,49,2
Up Type= 0
Dn Type= 2

--- 25_ras.g01 (geometry) ---

Geom Title=25
Program Version=4.10

River Reach=25,49
Reach XY= 30
1187241.22303113835834.547653437 1187334.5563325835676.214364186
1187360.38965484835557.8810650711187402.88964102835512.881077141
1187481.22294319835231.2144914271187523.72292861835157.881178543
1187671.94170344835016.9370859271187705.68695822834882.304395333
 1187763.4610002834824.5303533081187945.27930892 834756.56089215
1187984.36174905834722.5761615341188017.73686817834679.665294155
1188038.72276106834593.7146636551188132.88939577834446.214704528
1188251.22269452834451.2146996261188348.72266471834412.048041716
1188482.05595052834121.2147904341188574.55592111 834044.54814373
1188687.88921607833867.8815260231188748.72252676833703.714906096
1188817.88916373833380.3816662881188797.05965587833271.249434695
1188805.09299287833179.6693927051188871.36321756833060.722835645
1188959.72351706832992.7533744571188992.00901109832914.588494077
 1188915.5433673832754.860260308 1188915.5433673832705.582400948
1189024.55574754832612.8818870931189113.72238445832490.381920695

Type RM Length L Ch R = 1 ,4192.087,47.417700,47.417700,47.417700
XS GIS Cut Line= 6
1187384.07539079835880.6159778521187285.92473024835842.283271854
1187261.03517745835836.0406396951187223.23138134835831.501044355
1187196.50544193835825.8202697471187096.34808471835792.866793337
#Sta/Elev= 30
9849.036222.29539855.423220.7306 9860.06218.96279867.166217.34719913.331208.2471
9934.211202.99959944.651198.60359955.073193.1414 9978.75183.59959988.704178.4937
 9995.32174.37459998.628172.907610001.92173.176110025.15 182.24610048.69192.6307
10058.96197.522710072.65207.161610076.07 209.06810079.49209.917610101.42211.4538
 10103.7212.095310117.61219.152410121.09220.236810124.56220.479110128.04221.3335
10131.52224.416110134.99228.929210138.47 232.80410141.95234.781410150.97235.5368
#Mann= 3 , 0 , 0
9849.036    0.12       09849.036    0.12       010150.97    0.12       0
#XS Ineff= 2 , 0
       0                               0
Bank Sta=9849.036,10150.97
Exp/Cntr=0.3,0.1

Type RM Length L Ch R = 1 ,4144.669,47.417700,47.417700,47.417700
XS GIS Cut Line= 6
1187390.50485424835853.6860473421187294.86477979835809.342250385
1187255.08582702835789.2268108421187253.28681067835788.353002966
1187209.36429337835766.5576944931187116.67213868835726.555793567
#Sta/Elev= 30
9849.004206.38649856.462204.65999885.393199.46279889.009198.99519892.625198.9832
 9917.94194.67549931.205190.01419950.487 179.6339954.592177.92919965.127174.4138
9983.673165.97049998.215161.020310001.87160.4197   10013164.520810016.52166.1108
10031.17 175.94410056.65192.471610060.22193.747510063.79194.171910078.09194.5795
10081.66195.311910085.23  196.8310088.81199.8542 10103.1214.219810113.82224.3976
10117.39226.793110120.96228.251310124.54 228.93310131.68228.565110150.99234.5346
#Mann= 3 , 0 , 0
9849.004    0.12       09849.004    0.12       010150.99    0.12       0
#XS Ineff= 2 , 0
       0                               0
Bank Sta=9849.004,10150.99
Exp/Cntr=0.3,0.1

Type RM Length L Ch R = 1 ,4097.252,47.417700,47.417700,47.417700
XS GIS Cut Line= 6
1187411.54079129835825.3702444561187331.39011427835783.041899233
1187259.49480449835735.0028779031187230.27840963835717.390462526
1187190.23431548835696.6125754011187148.85372402835677.469717891
#Sta/Elev= 30
9849.047195.09149861.937190.36669876.778186.58489887.908182.19139902.749178.2386
9911.633174.75829925.684172.1021 9943.79169.64119967.364168.28759971.293 166.967
 9983.08159.53899990.938155.49879994.866154.08599998.795153.1584   10001153.0557
10005.08  153.7810010.88156.165210041.19171.715610045.81174.325310053.48179.4664
10057.31180.926810061.11182.105510079.59182.552610081.62183.266710112.69 203.333
10130.76210.970210141.83212.965310145.22213.923610148.84 216.05210150.98217.7306
#Mann= 3 , 0 , 0
9849.047    0.12       09849.047    0.12       010150.98    0.12       0
#XS Ineff= 2 , 0
       0                               0
Bank Sta=9849.047,10150.98
Exp/Cntr=0.3,0.1

Type RM Length L Ch R = 1 ,4049.834,47.417700,47.417700,47.417700
XS GIS Cut Line= 6
1187435.16020615835788.2806244111187355.02237664835744.540324892
1187323.62111203835723.382923551 1187292.2289921835698.760729222
1187269.13243628835684.2494222991187174.13153025835638.242225305
#Sta/Elev= 30
9849.025188.88519855.205184.94339862.591182.11369867.623181.39439892.138  180.63
9899.618 179.2659910.981   174.39933.707 159.2759945.281158.25669953.683158.4968
9965.061154.62419972.973154.70069981.025152.75119989.352149.83499998.581148.7367
10010.26149.9911 10022.4152.655810030.15155.228910045.39162.163810060.42170.9294
10064.12172.186610067.82173.1362 10086.3172.887710089.94174.854310097.16180.1245
10118.85191.450410129.69198.3107 10133.3199.950510144.15   201.210150.97202.8614
#Mann= 3 , 0 , 0
9849.025    0.12       09849.025    0.12       010150.97    0.12       0
#XS Ineff= 2 , 0
       0                               0
Bank Sta=9849.025,10150.97
Exp/Cntr=0.3,0.1

Type RM Length L Ch R = 1 ,4002.416,47.417700,47.417700,47.417700
XS GIS Cut Line= 6
1187473.44315489835734.6081682331187344.67658102 835676.37237095
1187336.62075764835673.1833661151187334.72339103835672.550910635
1187281.21958524835653.082856634 1187195.6326001 835616.56644043
#Sta/Elev= 30
9849.013180.65259858.918179.76639871.849177.45489886.252173.96739900.655169.4455
9907.856168.29889911.457167.28329929.461161.30179958.267150.15849965.468147.7859
 9972.67146.37669983.472 145.5299994.195143.10659997.724143.082610018.67144.4706
10036.12146.581510039.61147.648610042.54149.298910052.13156.935710057.07159.6976
10067.75162.685710082.02168.005310085.59168.267510092.72167.267410110.56166.6815
10114.12167.740310117.69169.368610124.82173.244310139.09181.861110150.99187.1264
#Mann= 3 , 0 , 0
9849.013    0.12       09849.013    0.12       010150.99    0.12       0
#XS Ineff= 2 , 0
       0                               0
Bank Sta=9849.013,10150.99
Exp/Cntr=0.3,0.1

Type RM Length L Ch R = 1 ,3954.999,47.417800,47.417800,47.417800
XS GIS Cut Line= 6
1187480.40139783835680.5905226351187409.57387311 835651.55731465
1187347.58963834835633.4297876591187323.88264688835621.807952717
1187264.34501469835600.3583055111187198.55223792835573.411254335
#Sta/Elev= 30
9849.062172.58459850.703171.61789871.978166.76979882.615163.18699889.707159.4793
9910.981146.41659918.073143.84759921.618143.16529928.599142.94589955.945139.6639
9969.618139.11889986.709139.43859990.127 139.14610001.08136.357210004.74135.8572
10019.23  137.2310034.62142.637310047.13146.117310050.62147.624510064.57 156.098
10075.03160.407810078.52161.016210082.04161.038110089.13160.278710106.86159.6681
 10110.4160.836910121.04169.141710124.58170.798310145.85173.219310150.98174.6057
#Mann= 3 , 0 , 0
9849.062    0.12       09849.062    0.12       010150.98    0.12       0
#XS Ineff= 2 , 0
       0                               0
Bank Sta=9849.062,10150.98
Exp/Cntr=0.3,0.1

Type RM Length L Ch R = 1 ,3907.581,47.417700,47.417700,47.417700
XS GIS Cut Line= 6
1187494.25844666835638.5172226031187390.14573963835594.211198862
1187369.94987883 835587.74188697 1187339.9231355835582.264515748
1187317.02377024835575.4438015521187212.28063784835532.606149999
#Sta/Elev= 30
9849.029165.16029855.042160.38759865.413 153.3919869.305151.4192 9872.87150.4294
9887.132150.58419901.395149.51679907.306147.47889915.684142.84079926.353 138.297
9944.181133.40769947.747132.92619954.878132.7642 9972.35133.71349975.795133.3285
9989.385 129.4679996.063128.856710009.39129.447610033.23131.9926 10052.8137.4357
10068.52141.1003 10082.7146.690510093.33151.536310096.87151.7217 10114.6150.8007
10118.14150.826810121.69151.541710125.23153.663110139.47165.248810150.97173.3091
#Mann= 3 , 0 , 0
9849.029  0.0941       09849.029  0.0941       010150.97  0.0941       0
#XS Ineff= 2 , 0
       0                               0
Bank Sta=9849.029,10150.97
Exp/Cntr=0.3,0.1

Type RM Length L Ch R = 1 ,3860.163,47.417700,47.417700,47.417700
XS GIS Cut Line= 6
1187505.62974424835617.3162114561187414.39749501835574.140959356
 1187389.1491872835557.7538319511187360.16985586835530.500074964
1187339.27529271835515.6190354671187244.63260574835469.362671723
#Sta/Elev= 30
9849.055158.73069860.414155.00669864.017154.19189878.429154.10629889.238152.5246
9896.444152.24479900.047151.16929907.253145.93499910.856144.25119925.522138.6677
9937.935135.22459947.599130.34089951.359 129.413 9955.27129.06319970.915129.5386
9974.827129.08149980.111127.43639991.942121.73219996.254120.7399    9999120.6925
10010.51122.319610027.21123.373410045.55125.318510083.51130.419810109.85135.8157
10114.53137.706510122.44142.087510127.87143.8638 10145.9145.024710150.95146.0789
#Mann= 3 , 0 , 0
9849.055   0.065       09849.055   0.065       010150.95   0.065       0
#XS Ineff= 2 , 0
       0                               0
Bank Sta=9849.055,10150.95
Exp/Cntr=0.3,0.1

Type RM Length L Ch R = 1 ,3812.745,47.417700,47.417700,47.417700
XS GIS Cut Line= 6
1187542.96092266835567.8070605941187418.48871224835513.193053758
1187405.32717268835508.2360732981187395.16312084 835504.55579313
1187327.58895379 835471.921805241187267.13183196835445.117321159
#Sta/Elev= 30
9849.009161.38499854.495 161.2389860.465 159.4559868.631155.66219876.796151.4143
9879.574150.17659883.157149.06259893.905148.28839897.488147.29199904.653144.1926
 9925.79138.0233 9940.48132.07899958.394121.96919961.977120.90549969.142120.3137
9987.011119.68279991.979117.98069997.528117.0494    9999117.030910004.49117.5482
10018.29117.996310033.38118.857810051.65120.763610073.51123.616110088.03125.0539
10109.57132.147810120.33 136.01510127.51138.213110134.86 140.05310150.99142.9296
#Mann= 3 , 0 , 0
9849.009   0.065       09849.009   0.065       010150.99   0.065       0
#XS Ineff= 2 , 0
       0                               0
Bank Sta=9849.009,10150.99
Exp/Cntr=0.3,0.1

Type RM Length L Ch R = 1 ,3765.328,47.417700,47.417700,47.417700
XS GIS Cut Line= 6
1187558.19592623835510.1808825791187459.52028931835473.147230475
1187433.17981874835465.6516187911187394.10537146835457.206073878
1187371.36189222835450.2710428181187273.31546763835411.568997931
#Sta/Elev= 30
9849.032145.40059860.157144.8899 9870.67143.81759875.535141.90529881.183138.7167
9898.704133.34729933.747125.67059947.764 123.1679951.268122.07829964.997116.6781
9968.408115.58949971.819115.1837 9992.11115.120310012.25115.614410022.34114.8193
10040.82115.317910056.95116.823410074.59117.6958 10088.7 117.67510092.23118.3375
10095.75120.167810099.28123.273110102.81126.869710106.33129.856810109.86132.1135
10113.39133.004910116.92132.943710131.02135.317610140.09139.001610150.98140.8703
#Mann= 3 , 0 , 0
9849.032   0.065       09849.032   0.065       010150.98   0.065       0
#XS Ineff= 2 , 0
       0                10053.52       0
Bank Sta=9849.032,10150.98
Exp/Cntr=0.3,0.1

Type RM Length L Ch R = 1 , 3717.91,47.417700,47.417700,47.417700
XS GIS Cut Line= 6
 1187571.6717434835471.771775059 1187459.7950918835429.640183567
1187431.75574419835417.7780412011187429.92914039835416.963474705
1187392.55273066 835401.312288741187289.95404532835363.132858338
#Sta/Elev= 30
9849.008145.44739878.043134.65969885.054 132.3579895.572130.97399927.124121.4593
9930.629120.53859937.641119.50429948.158116.81679951.664115.79739958.675112.8604
9962.181111.988410001.28108.450710004.84108.423910011.95109.664610015.51109.6825
10064.93108.081410071.93108.145810078.93108.785610082.43109.552710089.43111.7457
10092.93112.282810110.44112.226110113.94112.629210117.44114.188510120.94 116.273
10127.94117.789210138.44122.947610145.44127.088310148.94128.495610150.99128.9612
#Mann= 3 , 0 , 0
9849.008  0.0582       09849.008  0.0582       010150.99  0.0582       0
#XS Ineff= 2 , 0
       0                10039.93       0
Bank Sta=9849.008,10150.99
Exp/Cntr=0.3,0.1

Type RM Length L Ch R = 1 ,3670.492,47.417700,47.417700,47.417700
XS GIS Cut Line= 6
 1187591.7097057835422.327760102 1187518.2286512835395.592421931
1187449.80609234 835373.861054761187447.88119298835373.318134483
1187372.85471146835349.6433111321187305.41115887835326.451304258
#Sta/Elev= 30
9849.016136.94399857.359133.44279864.341131.46699867.832130.81099878.306 129.882
9892.271127.44069909.727123.42139920.201120.38289940.953115.47429954.722110.1149
9961.607 108.2939965.049107.83959985.703107.29929989.146106.5006 9996.03103.6589
9999.468103.115510006.33104.815410013.22105.743310047.62106.223210075.14106.0648
10095.92106.496310099.39107.057510106.33109.3139 10109.8109.744910127.14110.0963
10130.61110.788810134.08117.396410137.55121.431910144.49123.939110150.99124.8063
#Mann= 3 , 0 , 0
9849.016   0.052       09849.016   0.052       010150.99   0.052       0
#XS Ineff= 2 , 0
       0                10040.83       0
Bank Sta=9849.016,10150.99
Exp/Cntr=0.3,0.1

Type RM Length L Ch R = 1 ,3623.075,47.417800,47.417800,47.417800
XS GIS Cut Line= 6
1187604.92658077835369.8390280271187563.02846587835353.756658946
1187525.01749776835341.824492802 1187401.4697358835315.494874049
1187359.56504868 835303.590694811187314.74993288835288.344507762
#Sta/Elev= 30
9849.034131.72919882.132124.6252 9896.14119.74679909.894 116.2659927.088113.6789
 9933.96112.30929940.679111.31529947.397109.92389967.552103.9273 9977.63103.4601
9991.066103.31969994.426 102.7859997.785101.573510001.14 99.933310004.49 99.4152
10011.19102.731210014.54103.697910041.34104.927810058.08105.303310085.33105.5175
10092.15105.821310098.97106.279810102.08106.7873 10109.3108.866210112.76109.4498
10126.62109.362210133.55109.550710137.02109.987110140.48111.839710150.98120.6503
#Mann= 3 , 0 , 0
9849.034   0.071       09849.034   0.071       010150.98   0.071       0
#XS Ineff= 2 , 0
       0                10038.68       0
Bank Sta=9849.034,10150.98
Exp/Cntr=0.3,0.1

Type RM Length L Ch R = 1 ,3575.657,47.417700,47.417700,47.417700
XS GIS Cut Line= 6
 1187608.5696531835326.9547779491187567.22719332835309.493466938
 1187535.8282247835298.3562656441187406.68494933835266.289112273
1187363.31408038835252.3508934711187321.06800197835236.509220852
#Sta/Elev= 30
9849.018119.98099854.462119.18139868.708119.05749886.516118.2042 9911.05118.1715
9921.493117.62029927.213116.95929931.842116.06139935.254114.78199952.311 104.661
9959.125101.25419962.487100.1264 9965.8599.791969986.026100.19689989.388100.0056
9999.47897.5390710002.8697.1935710006.2397.6700310016.37101.264810019.75 101.678
 10026.5102.266410050.15103.202910060.29104.389510074.07105.363810101.64 109.018
10112.08109.7565 10126.1110.1586 10133.1113.698110136.61114.520110150.98116.2369
#Mann= 3 , 0 , 0
9849.018   0.073       09849.018   0.073       010150.98   0.073       0
#XS Ineff= 2 , 0
       0                10033.37       0
Bank Sta=9849.018,10150.98
Exp/Cntr=0.3,0.1

Type RM Length L Ch R = 1 ,3528.239,47.417700,47.417700,47.417700
XS GIS Cut Line= 6
1187617.02657554835297.877933444 1187546.6542449835263.792430179
1187480.49582497835235.9162278841187478.62772128835235.201953006
1187413.40922626835207.9548412731187341.11027181835175.344324634
#Sta/Elev= 30
9849.016119.06479885.857119.22599896.794118.31359904.085117.20939917.719 117.176
9922.312116.54559925.957 115.3799929.547113.41629943.787104.59929958.02897.97556
9961.58897.408919986.50997.49204 9990.0797.2155510000.7393.7740310004.2894.10885
10011.3996.9035610014.9597.4118410022.0697.9327510035.25 97.590410046.9597.90901
10057.61100.133610068.2899.9033310086.23100.635510089.83101.516510093.43104.8229
10097.03 107.55510100.63108.332810133.02109.189410140.22 113.61110150.99114.0835
#Mann= 3 , 0 , 0
9849.016  0.0468       09849.016  0.0468       010150.99  0.0468       0
#XS Ineff= 2 , 0
       0                10020.61       0
Bank Sta=9849.016,10150.99
Exp/Cntr=0.3,0.1

Type RM Length L Ch R = 1 ,3480.821,47.417700,47.417700,47.417700
XS GIS Cut Line= 5
1187629.50023315835271.5998679811187501.36627388835193.618768832
1187499.69635744835192.5181421541187494.08469206835189.074970152
1187370.14572374835116.917820653
#Sta/Elev= 30
9849.002119.20169856.331118.62259875.534118.53859887.616116.40679906.549111.9542
  9910.1111.40829921.622 110.7289929.303108.78639933.144107.26889938.102104.7955
9948.50798.134579952.34796.118449956.18895.52384 9967.7195.162019983.07295.46595
9988.58894.733589994.59492.248629998.43591.6752610002.3291.7514810006.1792.24021
10009.9993.3222110013.79 93.490310055.5594.1154810059.3494.7964810066.0497.39777
10070.7398.45426 10097.3101.6726 10104.9102.051810139.06 105.753   10151105.3233
#Mann= 3 , 0 , 0
9849.002   0.045       09849.002   0.045       0   10151   0.045       0
#XS Ineff= 2 , 0
       0                10014.49       0
Bank Sta=9849.002,10151
Exp/Cntr=0.3,0.1

Type RM Length L Ch R = 1 ,3433.404,96.498900,96.498900,96.498900
XS GIS Cut Line= 6
1187717.93224111835300.0742513391187593.35909426835212.675603032
1187502.88193923835130.6681340491187461.22785777835097.636028931
1187405.88990471835060.4986471981187266.88430059834980.032720163
#Sta/Elev= 30
9759.942139.21279794.982133.26589829.298124.92959854.578120.03219883.146117.4236
9903.552107.5009 9912.96104.54759923.125103.69269928.207102.34439946.05894.69201
9963.24293.97293 9981.03 94.3423 10001.888.7132210013.1291.3202210044.0491.47759
10097.8589.8069310117.6190.1184610125.5191.6142510137.3696.36121   1015797.83278
10175.95 96.138110187.3392.57768 10198.791.4988710205.0791.7605210211.6192.74107
10221.4495.5146410247.9898.59762   10264103.490510283.65105.772110314.76113.5563
#Mann= 3 , 0 , 0
9759.942   0.045       09759.942   0.045       010314.76   0.045       0
#XS Ineff= 2 , 0
       0                10016.25       0
Bank Sta=9759.942,10314.76
Exp/Cntr=0.3,0.1

Type RM Length L Ch R = 1 ,3336.905,96.498800,96.498800,96.498800
XS GIS Cut Line= 6
1187871.15405528835314.6954408791187682.86310412  835175.2982855
1187634.58381194835129.4757261471187570.74747546835058.321564659
1187526.11164959835018.373081869 1187323.8555494834879.409649818
#Sta/Elev= 30
 9649.06 168.4349707.677147.69219747.924 137.2159775.117127.21239797.539128.3857
9804.664127.68139838.124119.84439854.855117.66899884.192110.27539910.888100.5388
9934.717 93.39519962.10292.836779984.22190.380299988.61289.4026710001.7483.43151
10019.4785.7801710067.5886.8034310138.4185.0308910184.3687.9556210188.4389.60347
10204.43   100.310208.36101.980710216.22103.500410229.43103.221210239.82105.0042
10259.18111.539410282.98123.276810302.74129.443810318.68 136.87910350.93145.0223
#Mann= 3 , 0 , 0
 9649.06   0.045       0 9649.06   0.045       010350.93   0.045       0
#XS Ineff= 2 , 0
       0                10027.68       0
Bank Sta=9649.06,10350.93
Exp/Cntr=0.3,0.1

Type RM Length L Ch R = 1 ,3240.406,96.498900,96.498900,96.498900
XS GIS Cut Line= 6
1187952.49931319835226.6642016851187836.93245305835136.280210827
1187756.57931628835078.5339554721187658.06891684835015.573930024
1187532.68508126834944.8767318961187369.47097032 834837.57696844
#Sta/Elev= 30
9649.038155.28049747.147124.12129762.988121.93639775.483115.00229789.752113.5067
9800.662110.96829811.905106.61769820.533 104.7269834.393103.22199889.21693.60818
9966.61888.08007 10080.983.5305210118.96 83.704910133.4585.3630510146.2585.34378
10170.7789.3809210180.7792.4554110192.5599.6638210206.61106.333410220.03108.2315
 10230.5113.382610247.52113.921910255.37115.914110284.25134.487310290.22136.9862
10320.08 139.28810326.06141.254210332.03147.3013   10338149.732210350.97 150.184
#Mann= 3 , 0 , 0
9649.038  0.0825       09649.038  0.0825       010350.97  0.0825       0
#XS Ineff= 2 , 0
       0                10032.75       0
Bank Sta=9649.038,10350.97
Exp/Cntr=0.3,0.1

Type RM Length L Ch R = 1 ,3143.907,204.347800,204.347800,204.347800
XS GIS Cut Line= 6
1187884.28881449 835130.857372941187786.01610282834967.897137001
1187732.00685284834940.7684421241187648.02898532834918.320391178
1187590.09172225834892.5801386091187384.79751009834757.156373456
#Sta/Elev= 30
9703.625116.39769731.288112.57599742.782107.86769754.276106.5085  9769.6100.7144
9811.74491.562499838.56389.984279869.21282.178069915.02982.532779951.403 74.3491
9972.20272.409529989.15472.9960810010.1470.0784110022.8270.4816110054.2676.26096
 10104.9 88.767310112.0891.5449710123.4598.4685910134.82102.301310178.76113.2301
10196.72115.579710200.64 125.65910204.63130.124110212.61132.240810231.71132.8664
10243.24141.328710260.48145.544610316.34172.602810341.25177.818210350.96182.1068
#Mann= 3 , 0 , 0
9703.625  0.0663       09703.625  0.0663       010350.96  0.0663       0
#XS Ineff= 2 , 0
       09924.692        10030.39       0
Bank Sta=9703.625,10350.96
Exp/Cntr=0.3,0.1

Type RM Length L Ch R = 1 ,2939.559,41.393500,41.393500,41.393500
XS GIS Cut Line= 6
1187939.13763803835166.2201604791187850.77733853834885.846133123
1187841.24636441834830.9912923231187809.58075499834735.994464094
 1187770.9379774834696.8149812771187597.59109562834581.682794327
#Sta/Elev= 30
9617.002136.81579630.758132.55989644.518123.28479663.783121.95089692.677113.1766
9706.436112.13259713.316110.85749727.076105.11859747.715101.98229785.55490.52893
9802.75388.437469826.83386.870079840.59281.724329861.23277.459249922.76177.31419
10007.1978.6793510100.2678.8075310126.2778.1124310157.7880.9050710173.5384.33824
10185.3588.5136510205.0499.2056910210.76101.525510234.48106.515510252.27112.8342
10268.05123.005810299.71141.022410315.32 152.69310323.19156.213710330.35156.5621
#Mann= 3 , 0 , 0
9617.002  0.0479       09617.002  0.0479       010330.35  0.0479       0
#XS Ineff= 2 , 0
       09955.489        10070.61       0
Bank Sta=9617.002,10330.35
Exp/Cntr=0.3,0.1

Type RM Length L Ch R = 1 ,2898.166,68.846400,68.846400,68.846400
XS GIS Cut Line= 6
1187966.26437414835141.2635632571187875.60825893834795.570914611
1187859.33221725834761.9337618351187826.78013393834709.850428507
1187737.03834943834631.3263670591187624.71783173834556.726197105
#Sta/Elev= 30
9629.762 135.0479641.431133.61249644.871132.28439648.311128.76059651.751126.8855
 9686.15113.7355 9703.35109.99739730.869 105.5179751.50897.523129761.82894.65544
9772.14894.418049806.54785.594989835.38984.299369850.80980.230789874.62976.58462
 9908.06 76.17289924.69176.659029941.32178.651089998.828 79.687710160.8778.25604
10175.7680.7882310195.7585.9071710220.3598.5104710235.27102.370910275.49119.3212
10287.31126.2856   10307139.507210326.69149.902410338.51159.284510340.67160.2907
#Mann= 3 , 0 , 0
9629.762    0.12       09629.762    0.12       010340.67    0.12       0
#XS Ineff= 2 , 0
       09957.905        10073.37       0
Bank Sta=9629.762,10340.67
Exp/Cntr=0.3,0.1

Type RM Length L Ch R = 1 ,2829.319,76.647300,76.647300,76.647300
XS GIS Cut Line= 4
1188009.07180062835010.4146646261187941.79749507 834779.29487294
1187917.92596725834715.275775731 1187721.5283978834537.324386835
#Sta/Elev= 30
9739.213102.5739 9744.37101.65859747.78799.809589758.03889.485739771.70688.52248
9792.20882.608079805.87680.191369840.04676.542359863.668 74.87179874.21675.17584
9891.30171.644449922.05471.121619976.726 64.11349987.15263.6330510025.6765.60671
10055.8365.0507210114.4665.8989510127.1567.3774310140.4370.0390510149.28 72.8774
10158.1477.3700710162.5678.3283910189.1376.7977110197.9877.3823610220.1286.80984
10242.2692.4771810264.39 101.66710295.25121.514510304.24 124.39610313.28 129.326
#Mann= 3 , 0 , 0
9739.213    0.12       09739.213    0.12       010313.28    0.12       0
#XS Ineff= 2 , 0
       0                10046.43       0
Bank Sta=9739.213,10313.28
Exp/Cntr=0.3,0.1

Type RM Length L Ch R = 1 ,2752.672,99.118600,99.118600,99.118600
XS GIS Cut Line= 6
1188248.88411598834951.5405019171188127.71905236834832.479598318
1188070.62267643834778.6844211351188012.97398962834728.247280183
1187894.54280057834630.3546310741187730.52814133834478.674989356
#Sta/Elev= 30
 9649.01118.03159666.014115.79459679.813108.71449712.505106.00769744.209107.7861
9763.996104.97199787.40199.023029804.00592.79878 9824.9887.911599862.902 82.5992
9880.93378.353169898.90976.514229929.42468.43426 9955.5863.336179989.968 63.0685
10011.1661.5447710041.0164.8767710095.0465.3175210117.7566.7651110148.5570.77954
10179.8477.2680310188.7977.2943910193.2478.3535810220.05 91.0759 10242.498.58637
10264.74 103.51410282.62116.730610287.08118.826310314.42126.046310350.98138.9403
#Mann= 3 , 0 , 0
 9649.01  0.1152       0 9649.01  0.1152       010350.98  0.1152       0
#XS Ineff= 2 , 0
       0                10046.38       0
Bank Sta=9649.01,10350.98
Exp/Cntr=0.3,0.1

Type RM Length L Ch R = 1 ,2653.553,60.164400,60.164400,60.164400
XS GIS Cut Line= 6
1188307.99433491834825.7685962261188141.14195405834674.248113285
 1188084.8377816 834641.671557611187985.15287045834608.420544722
1187932.12054189834581.1702796721187741.66852337834425.373745048
#Sta/Elev= 30
9649.063102.85639661.465102.32439697.27193.955559739.68594.084569763.24992.23626
9786.86193.358169819.68988.709969828.38286.217919845.25284.466679853.49284.92594
9897.57778.966449912.75878.456239934.97173.847569963.41560.082269990.84359.57014
10004.6157.8293210039.1262.1949410064.0761.9360810071.2765.1623910125.8964.93593
10141.0771.3753610157.2272.5354110186.3791.1802210227.16105.605110268.61122.3804
10292.01134.502110312.16147.694110326.93153.444410336.91 160.66810350.94164.3555
#Mann= 3 , 0 , 0
9649.063    0.12       09649.063    0.12       010350.94    0.12       0
#XS Ineff= 2 , 0
       09939.588        10040.86       0
Bank Sta=9649.063,10350.94
Exp/Cntr=0.3,0.1

Type RM Length L Ch R = 1 ,2593.389,56.288700,56.288700,56.288700
XS GIS Cut Line= 4
1188183.76798117834679.4684840741188086.11173114 834583.98237294
1187908.16034228834498.2618868351187774.69680062834384.329595163
#Sta/Elev= 30
9827.94578.737789845.01279.627659863.78378.980139877.86175.055689891.49373.38209
 9900.6774.845079905.25974.273259914.43669.05422 9932.79 63.19919943.56158.83505
9948.25458.060299972.11458.520019983.03854.898639997.605 57.089810030.3859.94407
10037.6660.0758910055.8758.6557510070.4458.7884210095.9360.1150810117.7862.94649
10127.3168.2554710194.41100.259910204.51106.034110243.33124.978210260.59131.3586
10269.22136.678810282.16146.938410286.47149.7178 10295.1151.169310337.53163.0765
#Mann= 3 , 0 , 0
9827.945    0.12       09827.945    0.12       010337.53    0.12       0
#XS Ineff= 2 , 0
       0 9965.73        10040.34       0
Bank Sta=9827.945,10337.53
Exp/Cntr=0.3,0.1

Type RM Length L Ch R = 1 ,  2537.1,92.259100,92.259100,92.259100
XS GIS Cut Line= 6
1188346.31177916834770.7654304421188230.30559365834650.541903602
1188174.12569129834596.7185868391188075.10113291834512.583621951
1187953.82716123834420.3482291191187822.38250636 834305.24525792
#Sta/Elev= 30
9643.33495.32135 9654.6490.372669677.36584.065789709.27979.863629736.63377.63186
9772.76271.433259782.21270.476179795.90270.326799819.03266.154699847.48666.48607
9856.971 65.87569871.19961.037039895.49761.165779904.83156.298059910.96854.63326
9926.43954.412189960.11355.650829995.30451.0012210002.1450.67678 10033.451.01922
10049.9552.7938610074.2452.9953610098.7557.6632410115.0962.3556810140.21 71.5045
10195.69 97.206410295.99 141.517 10317.8152.474210330.88156.940910345.27163.4061
#Mann= 3 , 0 , 0
9643.334    0.12       09643.334    0.12       010345.27    0.12       0
#XS Ineff= 2 , 0
       09958.789        10095.02       0
Bank Sta=9643.334,10345.27
Exp/Cntr=0.3,0.1

Type RM Length L Ch R = 1 ,2444.841,146.158900,146.158900,146.158900
XS GIS Cut Line= 6
1188345.40278453834723.2095003441188240.79065132834598.874824511
1188152.45178543834457.8147170061188097.32467876834417.977798946
1187972.02631847834284.4596082981187885.56924636834199.511318665
#Sta/Elev= 30
  9648.889.356279657.46185.876529673.99880.336629692.64970.273469697.04868.56104
9714.64265.64337 9748.7758.676429765.13859.015379824.323 53.07549874.55850.40067
9893.515 50.65129904.88952.155529920.05451.970499979.23349.4359310001.8247.76031
10031.17 50.105810058.2751.6000410063.9852.7297410077.4756.5710710082.2457.31564
 10115.857.6946110144.9657.1402610149.4658.4908510221.2896.7380310230.8199.85721
10239.85103.6315 10267.6111.966910286.67118.6157 10304.4123.071210350.58137.8428
#Mann= 3 , 0 , 0
  9648.8  0.0675       0  9648.8  0.0675       010350.58  0.0675       0
#XS Ineff= 2 , 0
       09869.495                       0
Bank Sta=9648.8,10350.58
Exp/Cntr=0.3,0.1

Type RM Length L Ch R = 1 ,2298.682,139.493200,139.493200,139.493200
XS GIS Cut Line= 6
1188492.04615528834712.3682781461188406.53038145834627.072816619
1188342.25654343834551.3184044721188298.69747527834486.566069552
1188204.76246957834317.6248436691188068.59597074834157.879248362
#Sta/Elev= 30
9655.44594.863579668.47993.694179691.05386.294359709.63781.703899770.03269.33317
 9794.7663.775089805.45760.27471 9827.3856.088039860.66952.07108 9882.1350.92042
9914.23147.354389945.30746.762659956.82445.7312810012.2445.1023410097.7147.38986
10148.6246.7781510159.68 45.117310168.9646.0072610170.7846.9429910176.3355.93985
10181.8856.8566510223.0356.2427710227.2655.73478 10235.753.1661810270.5853.55224
10274.9754.2144810283.7759.1313110296.9763.4473410346.6769.3702510357.3571.93906
#Mann= 3 , 0 , 0
9655.445  0.0632       09655.445  0.0632       010357.35  0.0632       0
#XS Ineff= 2 , 0
       0                               0
Bank Sta=9655.445,10357.35
Exp/Cntr=0.3,0.1

Type RM Length L Ch R = 1 ,2159.189,100.347400,100.347400,100.347400
XS GIS Cut Line= 6
1188663.23273031 834552.992364221188475.66312765834416.097737908
 1188328.6704975834333.3095142121188297.35337217834312.120802808
1188247.59728142834267.3889473151188110.34325105834127.245482351
#Sta/Elev= 30
9658.211 74.73389669.62769.965299680.56867.838219703.27260.796159711.47259.37452
9724.33257.922889740.17156.808269779.03856.74229 9795.4556.264629813.70554.14476
 9829.7153.210529845.71649.283049849.71748.947099873.72547.932249899.01546.03998
9916.67746.45405 9930.4646.03419 9973.62 43.24869988.50541.4262210008.1941.33368
10140.3543.6929610174.7843.6332210200.8745.0131210210.0645.8024110228.4248.74558
10265.1653.2865410288.1255.2619710311.0858.3870510329.45 60.070610360.1365.75921
#Mann= 3 , 0 , 0
9658.211  0.0497       09658.211  0.0497       010360.13  0.0497       0
#XS Ineff= 2 , 0
       0                               0
Bank Sta=9658.211,10360.13
Exp/Cntr=0.3,0.1

Type RM Length L Ch R = 1 ,2058.842,99.118700,99.118700,99.118700
XS GIS Cut Line= 6
1188716.72934124 834436.524780791188532.83719719834321.679432884
1188360.48185853834244.2285938071188306.52880334834214.412911501
1188234.98838415834161.2026668161188125.30589723834066.124405564
#Sta/Elev= 30
9649.04159.954129693.33452.422199712.93950.912819728.62450.286459740.38749.38759
9759.99248.725339804.67947.973989825.05145.399539874.13143.960579885.10443.08006
9910.70841.943449953.87539.269079993.01739.2117310003.7438.35481 10010.939.33029
10021.6539.8487410094.6940.1525110121.7441.3053110153.5641.0502810170.1842.64465
 10182.742.6607710186.8843.1632510198.75  45.63110209.1747.0823810238.2149.85665
10251.2450.5014410264.2652.0068210309.3458.9571610329.3863.4076410350.9769.04671
#Mann= 3 , 0 , 0
9649.041  0.0556       09649.041  0.0556       010350.97  0.0556       0
#XS Ineff= 2 , 0
       0                               0
Bank Sta=9649.041,10350.97
Exp/Cntr=0.3,0.1

Type RM Length L Ch R = 1 ,1959.723,99.118600,99.118600,99.118600
XS GIS Cut Line= 6
1188756.42054885834364.2942977561188577.79672266834250.931563378
1188458.94297169834179.9607308941188358.08036516834119.486849949
1188284.90339803834068.4850787611188169.53813114833980.369116495
#Sta/Elev= 30
9649.00977.870189666.08477.380649697.17172.886249725.98270.031359756.596 64.3519
    977160.083649778.772 58.94529793.33258.278879811.70154.455519836.19251.10758
9892.68548.151859936.80143.797879952.08643.550239956.67842.51049 9963.5538.91852
9967.37138.184839988.67537.90518 10005.636.5610110009.4236.8318410017.0739.05241
10043.8539.82689 10112.739.1898210150.7739.6603510156.5139.0683510168.5141.73036
10240.4450.9029910274.6456.5465810294.4960.5193710332.4469.5223510350.9775.28764
#Mann= 3 , 0 , 0
9649.009  0.0509       09649.009  0.0509       010350.97  0.0509       0
#XS Ineff= 2 , 0
       0                               0
Bank Sta=9649.009,10350.97
Exp/Cntr=0.3,0.1

Type RM Length L Ch R = 1 ,1860.604,99.118600,99.118600,99.118600
XS GIS Cut Line= 6
1188791.71350553 834308.860010351188573.07420997834161.748713828
1188533.37991193834126.8536658151188482.06271281834065.446784522
1188437.80205992834024.196333248 1188240.7793298833878.905986772
#Sta/Elev= 30
9649.081 91.5709 9673.1485.555289692.69477.554769723.98276.813269797.81261.68549
9810.02256.548079813.93355.821139829.82955.820279841.95952.221059866.21948.08514
9912.67641.958269949.85135.931279983.60634.2732810005.0235.0955910023.7933.78049
10044.3734.37722 10057.533.5852210067.1334.1747310100.8133.2451910136.3534.92542
10144.6738.6699810148.2639.5724110169.5940.2514610196.2746.0931110227.1454.49209
10258.0562.14686 10269.463.68206 10291.569.7925510311.6176.2721310350.9291.12145
#Mann= 3 , 0 , 0
9649.081   0.057       09649.081   0.057       010350.92   0.057       0
#XS Ineff= 2 , 0
       0                               0
Bank Sta=9649.081,10350.92
Exp/Cntr=0.3,0.1

Type RM Length L Ch R = 1 ,1761.486,99.118700,99.118700,99.118700
XS GIS Cut Line= 6
1188876.83119969834221.5475433021188750.99832925834144.075897161
1188608.41886417834048.2897368551188561.09956717834019.658014177
1188414.88643468833911.3758894151188294.14287497833830.823154541
#Sta/Elev= 30
9649.024113.11219680.214105.31239707.18393.777229711.99292.74431  9730.392.58978
9738.00591.336939745.71188.141459757.26981.279269762.05579.267089768.82877.97251
9795.79775.863439811.58172.090969823.43867.58959  9846.563.83398 9874.8256.92762
9878.77355.146699905.33353.999549926.20251.123089992.66231.9103510011.81 31.4055
10043.7133.2460810104.9532.36324   1012635.2174110137.0235.4811310175.6133.79407
 10186.635.2428910206.9741.3143410242.4754.4678110327.1379.5374510350.9687.57466
#Mann= 3 , 0 , 0
9649.024    0.12       09649.024    0.12       010350.96    0.12       0
#XS Ineff= 2 , 0
       0                               0
Bank Sta=9649.024,10350.96
Exp/Cntr=0.3,0.1

Type RM Length L Ch R = 1 ,1662.367,99.118600,99.118600,99.118600
XS GIS Cut Line= 6
 1188932.5200568834128.8058247911188735.53884094834015.365461451
 1188669.6387626 833973.413586121188595.45195517833920.522437059
1188526.43272307833875.1343261741188334.72467996833761.643604998
#Sta/Elev= 30
9649.017130.5186 9653.04129.12059671.853118.27889701.954105.14539705.717104.2484
9717.005104.11819747.10591.859019754.63190.202359765.91889.258619781.13381.61796
9784.94580.628749807.82379.029179861.20366.535649876.45761.408699889.89254.68294
9895.90353.61258 9911.4653.103259927.01746.306049968.29234.238339998.40929.26664
10062.5829.0936810117.5530.1382810144.7128.8313210163.9530.5525210187.0436.93572
10206.28 43.011610244.4757.8062310293.68 74.352210342.8989.6810710350.9893.02755
#Mann= 3 , 0 , 0
9649.017  0.1033       09649.017  0.1033       010350.98  0.1033       0
#XS Ineff= 2 , 0
       0                               0
Bank Sta=9649.017,10350.98
Exp/Cntr=0.3,0.1

Type RM Length L Ch R = 1 ,1563.248,99.118600,99.118600,99.118600
XS GIS Cut Line= 6
1189003.76124169834020.6309437321188801.46905552833922.222728786
1188689.71696602833866.1375628791188687.87630416833865.355281651
1188537.14459176833788.305077301 1188375.1315426833708.255726826
#Sta/Elev= 30
9649.005131.05319655.513129.71069673.756122.34799702.943120.21279724.834113.1661
9754.02198.625029764.96788.354099801.45182.712919812.39677.378749820.17376.07185
9830.63971.425349880.01954.657589889.10650.049439900.11942.003439903.78940.47698
 9916.5938.884319933.15639.24662 9951.5132.329939980.87730.309149991.889 26.7386
9999.22426.3496910124.44 28.119810150.2330.3007910190.6331.3279810216.2442.35401
10263.8159.5618310282.1162.6178610304.0770.9826210315.0572.7304210350.9981.92185
#Mann= 3 , 0 , 0
9649.005  0.1018       09649.005  0.1018       010350.99  0.1018       0
#XS Ineff= 2 , 0
       0                               0
Bank Sta=9649.005,10350.99
Exp/Cntr=0.3,0.1

Type RM Length L Ch R = 1 , 1464.13,99.118600,99.118600,99.118600
XS GIS Cut Line= 6
1189052.65310429833896.0519179181188841.39367548833813.637201866
1188759.99918852833784.6665343791188671.73551982833756.152379181
 1188590.9255848833726.8296005131188395.92770705833648.674317155
#Sta/Elev= 30
9649.008127.33139662.036121.63219690.311115.91539718.587106.49339768.04692.86699
9789.09884.51935 9810.1583.294499841.72877.392869852.25470.80417 9862.7861.23365
9887.25553.01697 9894.2249.51903 9908.1540.119169922.07934.313169956.90427.83517
    999923.7098310029.3425.2977210053.4924.8521210098.8526.0899910112.8124.85039
10126.7726.0085410151.2925.3540210200.5828.2720510235.7936.9281310264.0838.95487
10294.6849.7100710306.6851.9601410329.0761.8695510345.7273.6704110350.9976.45216
#Mann= 3 , 0 , 0
9649.008  0.1023       09649.008  0.1023       010350.99  0.1023       0
#XS Ineff= 2 , 0
       0                               0
Bank Sta=9649.008,10350.99
Exp/Cntr=0.3,0.1

Type RM Length L Ch R = 1 ,1365.011,99.118700,99.118700,99.118700
XS GIS Cut Line= 6
1189090.28732895833774.834079301 1188875.6720316833707.247431723
1188793.75936577833686.7625653521188688.18187948833665.230767582
1188587.51720301833639.0542019651188415.63328004833583.380404826
#Sta/Elev= 30
9649.024118.54299704.936100.73199756.84481.606439767.13481.258269791.08168.20198
9825.29145.649839831.25842.581499835.55441.300889845.81740.469769883.34141.85956
9910.39641.124869920.541 38.24729950.97825.843219957.74223.924459964.43923.94664
9974.472 22.580110028.0322.0276510054.8422.3732810078.4423.6673410115.7322.44835
10153.0224.0985510187.1126.6921310252.2735.1655910276.5340.7515410295.4942.74494
10307.7247.6366210311.1948.3843910325.0550.0054310335.4550.1123410350.9752.40668
#Mann= 3 , 0 , 0
9649.024   0.101       09649.024   0.101       010350.97   0.101       0
#XS Ineff= 2 , 0
       0                               0
Bank Sta=9649.024,10350.97
Exp/Cntr=0.3,0.1

Type RM Length L Ch R = 1 ,1265.893,99.118600,99.118600,99.118600
XS GIS Cut Line= 6
 1189109.2166615 833658.338834571188892.00108646833599.996313958
 1188812.9605299833585.1567508791188726.24510136 833577.56324175
1188640.83653877833562.9645626411188425.12552275833507.546861707
#Sta/Elev= 30
9649.064107.06689669.31996.90187 9682.9990.773099706.91377.293159720.58475.72917
9751.34361.990589781.86854.613779808.89540.236529866.32535.290379886.44630.55653
9899.79829.793869913.15128.172229939.85622.0231310019.1119.7455110042.1620.79379
10118.7120.6751310162.3925.1742210196.0730.0688410205.3232.6391610216.2833.49832
10229.7536.0657710236.49 36.6549 10246.639.9817910272.6443.9642310290.9353.18881
10297.7555.6083810314.8257.4486210332.2757.5481510345.5360.8209710350.9462.92517
#Mann= 3 , 0 , 0
9649.064    0.12       09649.064    0.12       010350.94    0.12       0
#XS Ineff= 2 , 0
       0                               0
Bank Sta=9649.064,10350.94
Exp/Cntr=0.3,0.1

Type RM Length L Ch R = 1 ,1166.774,99.118600,99.118600,99.118600
XS GIS Cut Line= 6
1189126.15456062833567.5704855241188999.01395116 833533.07429772
1188816.16778727833490.2156332381188707.12360135833467.324035354
1188541.33957621833435.149496073  1188441.992717833411.453845892
#Sta/Elev= 30
9649.013111.70159679.91298.683439737.70379.234879761.49968.068499785.25567.24671
9795.36565.803599802.10464.055819805.47462.000329812.21356.084829815.58353.92467
9839.17144.687339866.12936.559469886.348 28.70829933.52518.456629977.29719.01368
9997.43617.4231510030.9518.2159310044.3517.6461710084.5517.8208110134.6819.59921
10148.0522.6667410171.4426.5102810198.1833.4482810211.5540.1002110234.9446.50444
10255.0554.3135310282.0361.40163 10298.963.1487210322.5176.7091510350.9983.08559
#Mann= 3 , 0 , 0
9649.013    0.12       09649.013    0.12       010350.99    0.12       0
#XS Ineff= 2 , 0
       0                               0
Bank Sta=9649.013,10350.99
Exp/Cntr=0.3,0.1

Type RM Length L Ch R = 1 ,1067.655,99.118600,99.118600,99.118600
XS GIS Cut Line= 6
  1189156.214637833469.4755032621189035.87537255833436.929890598
1188847.98142829833398.3863617671188789.57793366833382.199649783
1188602.45831908833358.4093659271188468.86654112833332.235008461
#Sta/Elev= 30
9649.044107.81729663.494102.96589683.88694.273429721.27280.075989765.45560.54938
9768.85459.570579778.99159.714919809.24447.464559832.77439.13347 9856.2431.92106
9866.26829.886239899.69119.177519923.08816.145589936.45815.523179976.77117.59144
   1000115.7982110050.9516.3014610110.4815.3576710136.9317.4941310176.6228.31004
   1021343.2427810226.3147.4986110293.0276.4329810299.7378.0568110306.4483.34758
10319.8784.6852310326.58 91.791410329.9493.4356410346.7293.2609610350.9294.36138
#Mann= 3 , 0 , 0
9649.044    0.12       09649.044    0.12       010350.92    0.12       0
#XS Ineff= 2 , 0
       0                               0
Bank Sta=9649.044,10350.92
Exp/Cntr=0.3,0.1

Type RM Length L Ch R = 1 ,968.5368,99.118700,99.118700,99.118700
XS GIS Cut Line= 6
 1189145.4611295833338.0185455311188918.26181809833281.975627176
1188847.35826535833281.8701556831188766.91402813833303.137070252
1188698.86467376833306.9956286711188457.40634975833268.698628864
#Sta/Elev= 30
9649.08665.160329683.26754.225399696.975 54.16179720.96450.992439744.85940.43385
9768.61639.220559802.48929.591529815.90128.314139819.25326.911449829.31219.30599
9834.47217.78383  9852.716.312199872.58113.398529918.67412.830299958.16214.08278
10009.9913.4753810043.0914.67643 10056.313.8363210092.4614.5672710112.16 17.1361
10171.4636.3943710234.4565.7472310251.1572.6130310264.5176.7717810277.8782.67733
10291.2389.1304510308.0199.4688210314.74101.120910328.21101.607510350.93113.7819
#Mann= 3 , 0 , 0
9649.086    0.12       09649.086    0.12       010350.93    0.12       0
#XS Ineff= 2 , 0
       0                               0
Bank Sta=9649.086,10350.93
Exp/Cntr=0.3,0.1

Type RM Length L Ch R = 1 ,869.4181,124.606900,124.606900,124.606900
XS GIS Cut Line= 6
1189140.59013127833292.1077610071188982.05818667833240.045369965
1188881.91417444833211.4370115361188829.62968595833198.735047465
1188681.70505889833171.2436494071188462.33823997833114.676607785
#Sta/Elev= 30
9649.03547.451829664.53846.251479671.44444.205449702.52338.454869716.33634.80305
9743.96232.151089751.75229.325659778.49422.242769785.40121.657099802.66718.09162
9819.88516.017959864.24212.458499891.53912.683889949.23411.591599976.20112.22609
9996.08811.3173610032.5312.2511610052.6410.9783910082.86 12.924610113.0717.89457
10140.0224.6234110150.1529.6864410200.8148.9071710237.9664.0715410248.1468.58458
10265.1477.3299810312.7595.5132310329.75103.457710339.95105.675510350.97111.2164
#Mann= 3 , 0 , 0
9649.035  0.1158       09649.035  0.1158       010350.97  0.1158       0
#XS Ineff= 2 , 0
       0                               0
Bank Sta=9649.035,10350.97
Exp/Cntr=0.3,0.1

Type RM Length L Ch R = 1 ,744.8112,142.565600,142.565600,142.565600
XS GIS Cut Line= 4
 1189154.0917567 833184.070718851188856.72536403833083.815763588
1188742.87651652833051.5302695281188431.91623163832985.260044883
#Sta/Elev= 30
9687.762 48.45349689.85647.401049700.24345.810149710.629 40.45039731.403 33.8099
9745.25227.301829762.56427.081269790.26220.807349807.57318.665189850.41716.46037
9856.04515.11225 9862.9712.043779869.89410.932219928.75310.530629946.06411.41048
10038.979.18271110059.44 9.4646110069.6710.5667910090.139.14286910147.6410.19526
10161.0612.0064310167.7713.9534310204.6717.9151810234.86 24.732410252.7729.78518
10298.5949.6310510345.5665.1721610385.8173.0075810422.7178.1543910437.86 79.3312
#Mann= 3 , 0 , 0
9687.762  0.1075       09687.762  0.1075       010437.86  0.1075       0
#XS Ineff= 2 , 0
       0                               0
Bank Sta=9687.762,10437.86
Exp/Cntr=0.3,0.1

Type RM Length L Ch R = 1 ,602.2456,134.710500,134.710500,134.710500
XS GIS Cut Line= 6
1189481.82245205833196.3067606061189114.35308231833058.965950559
1189045.52198317833029.2714281811188869.14952604832946.275099232
1188594.72813949832867.5561107051188420.70796816832808.978229238
#Sta/Elev= 30
9439.354182.2278 9490.06173.53969507.548 165.9639539.027156.34579560.013144.8524
9584.496 123.438 9622.9798.623769629.96595.663299647.45493.183789664.94278.48662
9671.93774.700169713.909 71.80759727.90768.778449749.00353.737419766.58449.33491
9780.64841.420539794.71240.291829826.356 28.06899865.57517.379969904.87910.61514
9984.8557.17332910179.6210.4076810220.398.02044410237.379.94874610278.158.771098
10308.8511.0799710322.53  13.49210459.9221.7046510487.5422.0664510570.7428.39643
#Mann= 3 , 0 , 0
9439.354  0.0864       09439.354  0.0864       010570.74  0.0864       0
#XS Ineff= 2 , 0
       0                               0
Bank Sta=9439.354,10570.74
Exp/Cntr=0.3,0.1

Type RM Length L Ch R = 1 ,467.5351,196.347200,196.347200,196.347200
XS GIS Cut Line= 6
1189520.51669843832976.152271488  1189170.337178832860.044599463
1189058.59522264832848.9394984761188922.40063699832873.468505128
1188813.10825893832865.2323729541188494.42867503832726.997189188
#Sta/Elev= 30
9434.33150.38144 9463.4554.720049488.03451.287459523.15460.14494 9533.6960.40414
9613.80649.510889720.77422.821269741.33323.70002 9744.7122.626849748.08719.12289
9751.46417.544119758.21816.67364 9778.489.7481039858.572 6.562359954.026 6.11436
10074.478.40949510097.4410.7301910117.248.80997210192.237.90069910213.699.132957
10231.578.20346310260.188.93143410278.0610.43097 10331.79.81256710371.0412.87584
10388.9212.9964210474.7524.0363310491.73 27.680310506.9333.7223810512.1633.84797
#Mann= 3 , 0 , 0
9434.331  0.0867       09434.331  0.0867       010512.16  0.0867       0
#XS Ineff= 2 , 0
       09886.292                       0
Bank Sta=9434.331,10512.16
Exp/Cntr=0.3,0.1

Type RM Length L Ch R = 1 ,271.1879,131.140200,131.140200,131.140200
XS GIS Cut Line= 6
1189489.92170422832930.9392433051189003.00173139832751.795306536
1188962.48022655832722.7427692131188879.07557253832634.994103525
1188799.57866021832574.9175768911188432.26379245 832363.50924003
#Sta/Elev= 30
 9387.1537.724349418.75346.422569432.85254.847319450.47658.125839492.77549.96127
9531.54838.433859594.99525.845799622.94417.624879643.82616.509169664.7089.460379
9716.8645.9476069837.547 8.906329879.7224.74248810142.99 5.3120510186.948.262479
 10206.412.9808410221.9712.7750110225.8713.9308310253.1232.69494 10264.637.57875
10291.2941.6271110328.2251.1358710363.2853.8656610367.0356.0623110385.7776.30034
10408.2683.71513 10434.586.8350210463.4398.2272410486.97103.529810600.95122.2358
#Mann= 3 , 0 , 0
 9387.15  0.0852       0 9387.15  0.0852       010600.95  0.0852       0
#XS Ineff= 2 , 0
       09821.969        10164.14       0
Bank Sta=9387.15,10600.95
Exp/Cntr=0.3,0.1
